HEC-RAS study SHAVERN.prj: SHAVERN

--- SHAVERN.g01 (geometry) --- (continued)

Type RM Length L Ch R = 1 ,6764    ,147.2,148.9,149.8
XS GIS Cut Line= 4
2490229.76039546655267.9168423732490032.83867307655350.289327555
2489861.65835231655448.1066537092489777.99879704655486.718756138
#Sta/Elev= 30
       0 2261.11     7.6 2259.76    16.8 2256.26   29.67 2253.03    65.7 2245.04
   111.6 2239.74   121.7 2237.88     1542238.558   181.9 2236.98   206.3 2234.19
   238.9 2232.91  257.772230.495   275.8 2226.94   294.2 2226.48   321.8 2219.73
     331 2218.65   346.5 2218.73   354.1 2217.22   358.7 2217.62  360.722219.238
  363.212221.693  363.832222.588   377.1 2240.58   381.7 2245.78   386.3 2249.09
   420.9 2261.72     445 2277.62   451.1 2280.71   471.1 2288.41502.7531  2296.8
#Mann= 8 ,-1 , 0
       0      .1       0   29.67     .06       0     154    .055       0
  257.77      .1       0   346.5    .045       0  360.72      .1       0
  363.21      .1       0  363.83      .1       0
Bank Sta=346.5,360.72
XS Rating Curve= 0 ,0
Exp/Cntr(USF)=0,0
Exp/Cntr=0.3,0.1

Type RM Length L Ch R = 1 ,6615    ,100.2,99.3,98
XS GIS Cut Line= 4
2490161.54568117655132.774483872 2489956.9015383655246.036650997
 2489807.6014089 655302.667734562489718.79357332655372.169518932
#Sta/Elev= 30
       0 2295.07     7.8  2288.3    21.5  2265.8    26.1 2261.39    58.1 2253.17
  110.552243.827   122.1 2241.49   149.5 2240.15     192 2232.67  216.072233.365
   244.8 2230.47   273.5  2222.9   300.4 2219.28   315.3 2215.48     326 2216.93
   330.3 2215.95   338.9 2213.21   343.2  2213.8  346.582215.441   360.3 2220.43
   369.6 2225.08   375.8  2230.1   393.9 2247.55   399.7 2251.35  422.592258.545
   430.2 2261.73   442.8 2270.01   470.9 2283.04   485.5 2290.82506.3473 2297.19
#Mann= 6 ,-1 , 0
       0      .1       0  110.55     .06       0  216.07      .1       0
   330.3    .045       0  346.58      .1       0  422.59    .055       0
Bank Sta=330.3,346.58
XS Rating Curve= 0 ,0
Exp/Cntr(USF)=0,0
Exp/Cntr=0.3,0.1

Type RM Length L Ch R = 1 ,6516    ,140.3,139.7,138.7
XS GIS Cut Line= 4
2490130.65599923655046.5407884472489944.03083749655139.209834277
2489759.97981591655222.8693895392489684.04268113 655289.79703375
#Sta/Elev= 30
       0 2304.19    13.3  2298.3      49 2279.32    71.8 2269.48   122.5 2252.14
  152.292245.381   203.1 2234.81   215.1 2229.73   249.3 2228.89   253.7 2227.71
   266.9  2217.5   271.3 2215.78  298.462215.147   306.4 2215.11  310.042213.414
   317.8 2211.74     324 2211.84  330.572213.413     339 2215.07   381.3 2214.53
   385.5 2217.01   401.42240.614   407.5 2248.42   412.2 2251.69   440.8 2261.25
   460.2 2269.22   468.1 2273.23   477.1 2279.62   481.5 2281.87  511.76 2290.62
#Mann= 6 ,-1 , 0
       0      .1       0  152.29     .06       0  298.46      .1       0
  310.04    .045       0  330.57      .1       0   401.4    .055       0
Bank Sta=310.04,330.57
XS Rating Curve= 0 ,0
Exp/Cntr(USF)=0,0
Exp/Cntr=0.3,0.1

Type RM Length L Ch R = 1 ,6376    ,157.7,156.5,156.2
XS GIS Cut Line= 4
2490067.20644563 654920.609190732489846.51541666655024.775356406
2489673.49364995655120.1138809222489578.15512543655176.610784339
#Sta/Elev= 30
       0 2328.89    14.7 2322.18    20.1  2317.1      27 2307.63    47.1 2293.86
    70.9 2282.15   111.1 2264.79  150.042251.952   212.8  2233.8   227.4 2226.11
   252.9 2225.74     266  2220.9  283.652217.041  310.782211.015   316.8 2209.27
   333.8 2211.77   339.7 2212.84   362.5 2209.94   380.9  2212.9   408.2 2229.83
   439.1 2239.79   444.8 2242.82   454.4 2250.87  464.762264.974   471.9 2274.21
   477.3 2278.76   480.7 2280.07   495.9  2284.2   525.5 2288.03552.4103 2297.65
#Mann= 6 ,-1 , 0
       0      .1       0  150.04     .06       0  283.65      .1       0
  310.78    .045       0   333.8      .1       0  464.76    .055       0
Bank Sta=310.78,333.8
XS Rating Curve= 0 ,0
Exp/Cntr(USF)=0,0
Exp/Cntr=0.3,0.1

Type RM Length L Ch R = 1 ,6219    ,137.4,137.2,136.9
XS GIS Cut Line= 4
2489978.93003404654775.8358757252489786.48745678654869.408872009
2489620.52780299654985.9337353062489546.37561726655049.492751651
#Sta/Elev= 30
       0 2327.74    40.2 2310.59   83.762289.182   101.2 2281.77   153.3 2257.37
  187.462244.713   226.4 2230.26   232.1 2227.17   237.8 2222.77   240.7 2221.56
   263.7  2220.1   267.4 2218.86     278 2213.15  296.122208.641  299.79 2207.33
   311.4 2205.51   318.2 2207.19   321.1 2208.31   326.1 2208.56   344.1 2207.42
   355.8  2211.9   390.6  2218.8  406.492224.538   438.6 2239.94     449 2246.15
   458.4 2253.32   467.4 2264.26   471.8 2268.57   482.3 2270.77514.4326 2279.79
#Mann= 7 ,-1 , 0
       0      .1       0   83.76      .1       0  187.46     .06       0
  296.12      .1       0  299.79    .045       0   318.2      .1       0
  406.49    .055       0
Bank Sta=299.79,318.2
XS Rating Curve= 0 ,0
Exp/Cntr(USF)=0,0
Exp/Cntr=0.3,0.1

Type RM Length L Ch R = 1 ,6082    ,109.2,109.5,109.2
XS GIS Cut Line= 4
2489825.32907788654689.3249923672489685.85234757654777.601403956
2489541.07903256654883.5330978632489449.27156451654941.795529512
#Sta/Elev= 30
       0 2292.69    26.7 2278.82    45.42271.037    69.7 2261.86    78.8 2257.36
   107.6 2245.85  139.622233.989   153.8 2227.73   165.3 2219.07   188.2 2218.46
   201.1 2212.13   213.5  2208.9     235 2206.17   243.3 2204.29   258.1 2204.63
     268 2202.79   275.6 2204.63     297 2205.62   299.9 2206.55   302.7 2208.34
   311.3 2216.42   329.8 2228.75   360.2 2243.06   367.1 2247.67  374.952251.619
   389.9 2259.82   409.4 2267.62   432.8 2275.49   446.7  2276.7453.1895 2278.92
#Mann= 6 ,-1 , 0
       0      .1       0    45.4      .1       0  139.62     .06       0
   258.1    .045       0   275.6      .1       0  374.95    .055       0
Bank Sta=258.1,275.6
XS Rating Curve= 0 ,0
Exp/Cntr(USF)=0,0
Exp/Cntr=0.3,0.1

Type RM Length L Ch R = 1 ,5973    ,119.1,117.3,115.5
XS GIS Cut Line= 4
2489775.89428739654608.1106937052489625.82438769 654701.68368999
2489481.05107268654795.2566862742489403.36783048654849.988061459
#Sta/Elev= 30
       0 2289.77    24.9 2278.23    39.1  2272.4    76.8 2254.25  114.142239.117
   156.5 2223.64   166.3 2215.75   171.1  2213.7   180.5 2214.11   193.8 2213.28
     206 2206.89   213.9 2205.28  222.132204.329   226.52203.866   240.7 2201.93
   242.4 2202.09   247.2 2203.77   266.2  2203.6   280.5 2202.78   285.3 2203.72
   304.3 2212.53   328.2 2219.66   344.8 2225.39   356.4 2230.01   369.4 2237.74
   373.6 2241.47   382.2 2250.34   387.9 2253.42   419.5 2265.07444.2611 2271.22
#Mann= 5 ,-1 , 0
       0      .1       0  114.14     .06       0  222.13      .1       0
   226.5    .045       0   247.2      .1       0
Bank Sta=226.5,247.2
XS Rating Curve= 0 ,0
Exp/Cntr(USF)=0,0
Exp/Cntr=0.3,0.1

Type RM Length L Ch R = 1 ,5855    ,95.1,96.1,96.4
XS GIS Cut Line= 4
2489729.99055336654505.7100562622489564.03089958654590.455411388
2489451.03709274654689.3249923672489359.22962469654759.946121639
#Sta/Elev= 30
       0 2297.59     9.2 2291.55    26.1 2281.93      53 2268.82    66.5  2261.7
    99.3 2245.48   124.9 2234.77   175.7  2215.5  181.232212.747   188.1 2208.85
   213.1 2207.64   227.3 2203.53  243.892202.215   253.8 2200.65   266.9 2202.13
   273.1 2202.36   292.4 2201.29  301.392201.427     305 2202.06   306.6 2202.76
   315.6 2207.57   320.9 2209.98   345.6 2216.84   362.1 2222.35   382.3 2231.74
     392 2236.84   398.1  2241.1   403.4 2245.29   409.1 2248.35452.3146 2263.47
#Mann= 5 ,-1 , 0
       0      .1       0  181.23     .06       0  243.89    .045       0
   266.9     .06       0  301.39      .1       0
Bank Sta=243.89,266.9
XS Rating Curve= 0 ,0
Exp/Cntr(USF)=0,0
Exp/Cntr=0.3,0.1

Type RM Length L Ch R = 1 ,5759    ,103.4,102,100.4
XS GIS Cut Line= 4
2489682.32129111654428.0268140642489496.94082677654526.896395043
2489355.69856823654638.124673646 2489315.0914189654678.731822977
#Sta/Elev= 30
       0 2297.15    26.7 2281.28      63 2262.11    72.1 2258.41   103.8  2243.3
   135.5 2230.57  149.042224.389   167.6 2216.34   173.3 2214.49   180.9 2213.38
     194 2207.85     218 2207.38   223.1  2206.4   234.4 2202.77   253.6 2200.16
   262.9 2198.54     274 2200.66   294.4 2200.03   308.5 2200.95   314.7 2201.96
   325.6 2205.38   340.2 2211.72   345.9 2214.84   362.6 2226.03   388.3 2239.14
   402.3 2248.26   410.9 2255.82   416.6 2259.49   424.9 2262.62447.3058 2267.59
#Mann= 4 ,-1 , 0
       0      .1       0  149.04     .06       0   253.6    .045       0
     274      .1       0
Bank Sta=253.6,274
XS Rating Curve= 0 ,0
Exp/Cntr(USF)=0,0
Exp/Cntr=0.3,0.1

Type RM Length L Ch R = 1 ,5657    ,110.4,112.1,112.6
XS GIS Cut Line= 4
 2489648.7762547654316.7985354622489440.44392335654438.619983455
2489323.91906005654546.3172055932489258.59451548654593.986467851
#Sta/Elev= 30
       0 2318.94    12.1 2312.51    20.6 2306.35   28.312298.757    43.8 2290.14
    73.2 2275.71  134.762253.746   165.82241.965   206.2 2225.46   231.1 2217.09
   247.6  2207.9   270.9 2206.59   281.8 2201.79   299.3 2198.32   313.5 2199.53
     322 2198.22   327.6 2196.99     336 2198.27   347.1 2198.12   353.7 2198.67
  360.362199.994   367.3 2202.11   375.8 2205.57   412.7 2225.27   429.9 2237.95
   435.6 2244.39   441.3 2251.96     446 2255.98   468.8 2266.38480.8754 2270.24
#Mann= 7 ,-1 , 0
       0      .1       0   28.31      .1       0  134.76      .1       0
   165.8     .06       0     322    .045       0     336     .06       0
  360.36      .1       0
Bank Sta=322,336
XS Rating Curve= 0 ,0
Exp/Cntr(USF)=0,0
Exp/Cntr=0.3,0.1

Type RM Length L Ch R = 1 ,5545    ,91.6,93.1,94.4
XS GIS Cut Line= 4
2489569.32748427654253.2395191182489362.76068115654373.295438879
2489235.64264847 654473.930548092489179.14574505654516.303225653
#Sta/Elev= 30
       0 2298.78    44.6 2277.15   61.542270.401    90.9 2261.78  167.892236.196
   196.2 2227.72   231.3 2216.11   234.3 2214.82   240.1 2210.23   242.9 2208.95
   264.4 2208.98   273.7 2204.73  276.692203.951   279.8 2203.25     290 2198.89
   294.2 2197.66   308.4 2196.88   325.7 2197.24  328.852196.369   336.9 2194.32
     341 2194.71  346.182196.371   379.6 2215.48   383.3 2218.75   389.7 2227.23
   393.8 2231.93   420.7  2251.8   440.7 2261.21   462.7 2269.28471.6731 2274.06
#Mann= 6 ,-1 , 0
       0      .1       0   61.54      .1       0  167.89     .06       0
  276.69      .1       0  328.85    .045       0  346.18      .1       0
Bank Sta=328.85,346.18
XS Rating Curve= 0 ,0
Exp/Cntr(USF)=0,0
Exp/Cntr=0.3,0.1

Type RM Length L Ch R = 1 ,5452    ,103.7,103.3,102.6
XS GIS Cut Line= 4
2489451.03709274654226.7565956412489322.15353182654306.205366071
 2489198.5665556654378.5920235742489140.30412395654422.730229369
#Sta/Elev= 30
       0 2259.45    14.8 2255.06    32.3 2251.17   47.882246.513    89.6 2233.33
   102.1 2230.11   117.8 2224.35   145.1 2215.71   151.4 2213.17   160.2 2207.61
   164.6 2206.89   183.2 2206.31   192.4 2202.68   206.3 2199.58  216.212195.846
   221.6 2194.77   236.2 2194.39   243.4 2192.83   252.7 2194.42   266.6  2196.3
   275.9 2198.87   288.9 2204.26   308.4 2214.58   319.5 2222.47     329 2230.77
   337.5 2242.69   340.4 2245.82   343.3 2248.07   349.6 2251.43 367.723 2259.16
#Mann= 5 ,-1 , 0
       0      .1       0   47.88     .06       0  216.21      .1       0
   236.2    .045       0   252.7      .1       0
Bank Sta=236.2,252.7
XS Rating Curve= 0 ,0
Exp/Cntr(USF)=0,0
Exp/Cntr=0.3,0.1

Type RM Length L Ch R = 1 ,5349    ,141.1,140.5,139.9
XS GIS Cut Line= 4
2489371.58832231654150.8388816742489299.20166481654202.039200396
2489136.77306749654297.3777249122489071.44852291654339.750402475
#Sta/Elev= 30
       0 2245.39    15.7 2241.95    25.5 2239.15    52.3 2233.43   86.042223.818
    93.8 2222.05   101.3 2219.35   121.7 2213.52   126.3 2211.31   130.9 2207.73
   135.6 2206.09   158.8 2206.19   169.4 2202.08  192.662196.864   205.1 2193.56
   209.8 2193.05   218.2  2193.7   223.7 2192.09   228.3 2191.12   233.5 2191.97
   244.8 2193.08   250.4 2194.53     265 2200.28   279.6  2206.8   284.2 2210.15
   296.9 2224.42   303.3 2230.82     308 2234.48   312.8 2236.26 354.869 2246.48
#Mann= 5 ,-1 , 0
       0      .1       0   86.04     .06       0  192.66      .1       0
   223.7    .045       0   233.5      .1       0
Bank Sta=223.7,233.5
XS Rating Curve= 0 ,0
Exp/Cntr(USF)=0,0
Exp/Cntr=0.3,0.1

Type RM Length L Ch R = 1 ,5208    ,156.2,158.6,160.7
XS GIS Cut Line= 4
2489295.67060835654034.3140183772489157.95940627654113.762788807
2489036.13795827 654205.570256862488990.23422425654251.473990886
#Sta/Elev= 30
       0 2249.64   22.462241.876      45 2232.81    70.3 2223.48    89.2 2218.22
   105.2 2212.43   116.5 2208.97   124.1 2205.48   130.4 2201.67   132.9 2200.95
   158.1 2199.93     163 2198.78     173 2194.88     178 2194.19   187.4 2191.74
   200.7 2191.64   216.4 2190.81  233.962186.902   239.2 2185.37   243.2 2184.89
   247.8 2185.68  250.762186.904   253.5 2188.07   260.6 2192.29   273.5 2201.69
   278.2 2205.62   284.9 2209.44   341.7 2237.44   364.4 2246.74376.4455 2250.25
#Mann= 4 ,-1 , 0
       0      .1       0   22.46     .06       0  233.96    .045       0
  250.76      .1       0
Bank Sta=233.96,250.76
XS Rating Curve= 0 ,0
Exp/Cntr(USF)=0,0
Exp/Cntr=0.3,0.1

Type RM Length L Ch R = 1 ,5050    ,77.2,76.7,77.4
XS GIS Cut Line= 4
2489249.76687432 653928.382324472489101.46250285653988.410284351
2488977.87552662654043.1416595362488884.30253034654111.997260575
#Sta/Elev= 30
       0 2256.37    46.4 2238.46    81.3 2228.37   94.312223.858   105.6 2220.52
   145.6 2205.34     150 2203.01   154.3    2200   158.6 2195.95   160.9  2194.9
   185.2 2193.44   189.2 2192.18  196.452188.392   206.7 2185.05  237.632183.071
   241.7  2181.8   246.1 2181.47   254.8 2181.97  258.952183.071   263.6 2185.94
     268 2187.62   294.3 2191.75   313.9 2198.26   345.9 2207.02   358.6 2211.21
   363.6  2213.9   368.7 2219.39   373.5 2222.75   403.3 2234.73411.3328 2236.93
#Mann= 5 ,-1 , 0
       0      .1       0   94.31     .06       0  196.45      .1       0
  237.63    .045       0  258.95      .1       0
Bank Sta=237.63,258.95
XS Rating Curve= 0 ,0
Exp/Cntr(USF)=0,0
Exp/Cntr=0.3,0.1

Type RM Length L Ch R = 1 ,4973    ,113.4,109.6,108.2
XS GIS Cut Line= 4
2489205.62866852653873.6509492852489052.02771236653930.147852702
 2488931.9717926 653977.817114962488847.22643747654020.189792523
#Sta/Elev= 30
       0 2250.22    28.1  2239.2   58.212228.804    79.8 2221.81   113.9  2208.9
   122.4 2205.19   139.5 2199.15   143.7 2197.48   152.2 2191.98   155.9 2190.24
   169.3 2190.06   180.6  2189.2   186.8 2186.99   195.2 2185.37  203.922181.022
   208.1 2180.06   217.6 2179.52     221 2179.62  229.232181.023   251.1 2184.43
  261.062184.726   276.9 2186.41   289.9  2188.9   312.1 2195.34   342.3 2200.86
   356.8 2205.19   361.3 2207.42   370.2 2214.26   374.7 2218.77387.5833 2233.47
#Mann= 5 ,-1 , 0
       0      .1       0   58.21     .06       0  203.92    .045       0
  229.23     .06       0  261.06      .1       0
Bank Sta=203.92,229.23
XS Rating Curve= 0 ,0
Exp/Cntr(USF)=0,0
Exp/Cntr=0.3,0.1

Type RM Length L Ch R = 1 ,4864    ,152.6,154.5,156.7
XS GIS Cut Line= 4
2489142.06965218653751.8295012922489002.59292187  653818.9195741
2488875.47488918653907.1959856892488813.68140107653963.692889106
#Sta/Elev= 30
       0    2244    43.6 2228.24    74.7    2218    83.6 2216.14    96.9 2210.49
  118.07 2203.67   150.2 2194.01   160.4 2188.31   164.3 2186.76   183.8 2186.37
   188.7 2185.43   193.5 2183.16   197.8 2182.04   220.7  2180.5  225.852179.586
  228.022178.775   232.2 2177.44     238 2176.65  258.142178.774   266.7 2179.72
   273.9 2182.01   281.1 2183.37   298.3 2185.12   329.7 2193.21   352.3 2201.27
     358 2204.07   363.6 2208.01   369.3 2211.06   383.5 2216.27393.2647 2221.02
#Mann= 5 ,-1 , 0
       0      .1       0  118.07     .06       0  225.85      .1       0
  228.02    .045       0  258.14      .1       0
Bank Sta=228.02,258.14
XS Rating Curve= 0 ,0
Exp/Cntr(USF)=0,0
Exp/Cntr=0.3,0.1

Type RM Length L Ch R = 1 ,4709    ,126.5,127.3,128
XS GIS Cut Line= 4
2489127.94542633653605.2906580542488933.73732083653702.394710802
2488746.59132826653787.1400659282488683.03231192653815.388517636
#Sta/Elev= 30
       0 2267.19    28.9 2251.28    46.8    2242    59.5 2236.25    81.8 2227.67
  128.582214.092   154.1  2206.9   189.9 2198.27   200.4 2196.36   213.8  2191.7
   224.8 2184.61  232.46 2184.47   246.8 2183.79   255.5 2179.43   268.7 2176.75
   290.7  2176.2  301.422175.056   310.4 2173.08   313.5 2173.21  319.122175.054
   330.2  2178.2   347.8 2179.75   356.5 2182.65   378.5 2188.32   391.7 2192.77
   457.4 2217.69   461.4 2221.11   466.2 2226.48   470.6 2229.42492.1245  2238.6
#Mann= 5 ,-1 , 0
       0      .1       0  128.58     .06       0  232.46      .1       0
  301.42    .045       0  319.12      .1       0
Bank Sta=301.42,319.12
XS Rating Curve= 0 ,0
Exp/Cntr(USF)=0,0
Exp/Cntr=0.5,0.3

Type RM Length L Ch R = 1 ,4582    ,55.9,54.9,53.8
XS GIS Cut Line= 4
2489067.91746645 653511.717661772488875.47488918653598.228545127
2488720.10840478653652.9599203122488642.42516259653702.394710802
#Sta/Elev= 30
       0 2257.83    14.4 2249.22    33.5 2239.53    45.1 2234.21    66.8  2225.7
   81.212221.161   132.9 2205.88  184.032191.573   193.9 2187.69     203 2181.46
     206 2180.68   228.7 2180.03     233 2179.02   241.5  2175.8   254.2 2175.31
  268.372173.081   275.4 2171.23   279.6 2170.85   285.2 2171.22   291.52173.083
   296.6 2174.34   315.9 2173.47   345.4 2174.03     356 2174.96   360.2 2176.57
   369.5 2182.11   379.3 2185.73   405.8 2196.74   436.1 2207.74467.7971 2220.52
#Mann= 5 ,-1 , 0
       0      .1       0   81.21      .1       0  184.03     .06       0
  268.37    .045       0   291.5      .1       0
#XS Ineff= 2 , 0
          251.59 2176.58  305.92         2176.55
Permanent Ineff=
       F       F
Bank Sta=268.37,291.5
XS Rating Curve= 0 ,0
Exp/Cntr(USF)=0,0
Exp/Cntr=0.5,0.3

Type RM Length L Ch R = 1 ,4527    ,103.2,104.2,103.9
XS GIS Cut Line= 4
2489027.31031711653467.5794559752488864.88171979653536.435057015
2488716.57734832653603.5251298232488612.41118265 653640.60122269
#Sta/Elev= 30
       0 2249.54    44.1 2227.66    61.4 2220.77    85.3 2213.52     125 2203.08
     144 2197.17  149.022195.083   164.7 2189.51   174.4 2182.03   179.9 2178.93
   183.2 2178.41   196.3 2178.83   213.9 2178.21   227.1 2174.49  247.362172.318
   257.8 2170.47   262.2 2170.58   273.6 2172.44   294.8 2172.82   312.9 2171.93
     325 2173.37   337.7 2176.33  354.332177.502   368.3 2178.53   375.1 2180.24
   379.4 2182.66   392.1 2193.19   399.6 2197.38     443 2215.51449.7618  2217.4
#Mann= 5 ,-1 , 0
       0      .1       0  149.02     .06       0  247.36    .045       0
   273.6      .1       0  354.33    .055       0
#XS Ineff= 2 , 0
             217 2171.55     303         2171.55
Permanent Ineff=
       F       F
Bank Sta=247.36,273.6
XS Rating Curve= 0 ,0
Exp/Cntr(USF)=0,0
Exp/Cntr=0.5,0.3

Type RM Length L Ch R = 1 ,4423    ,152.4,150.5,149
XS GIS Cut Line= 4
2488986.78793251653381.3180231092488836.63326808653449.129807046
2488642.88531398653514.5197415562488546.01133693653570.222278361
#Sta/Elev= 30
       0  2252.2   19.922242.062    39.5 2231.68   51.742225.878    81.6  2211.7
      98  2207.4  122.78 2199.69   180.3 2183.57   183.6 2182.42   192.9 2177.02
   217.4 2176.68  224.352174.086   227.6 2172.91   233.9 2171.95   251.2 2170.39
  264.272169.976     275 2167.76   282.8  2169.8   293.9 2170.57   310.3 2169.35
   327.2 2172.13   356.7 2179.81   383.2 2190.01   387.9 2190.74   402.1 2191.33
  428.782203.318   443.2 2207.47   451.6 2210.55   466.3  2213.5480.9887 2218.46
#Mann= 8 ,-1 , 0
       0      .1       0   19.92      .1       0   51.74      .1       0
  122.78     .06       0  224.35    .055       0  264.27    .045       0
   282.8    .055       0  428.78      .1       0
Bank Sta=264.27,282.8
XS Rating Curve= 0 ,0
Exp/Cntr(USF)=0,0
Exp/Cntr=0.5,0.3

Type RM Length L Ch R = 1 ,4272    ,180.9,179,174.5
XS GIS Cut Line= 4
2488923.81984743653204.5230149892488739.75929103 653308.66254032
2488596.87017488653388.583571388 2488507.2617461 653446.70795762
#Sta/Elev= 30
       0 2270.79      15 2263.33    24.2 2256.78    55.4    2238    97.7 2216.57
   120.7  2206.7   146.3  2197.3  196.172181.329   205.1 2178.51   212.6 2174.39
   217.2 2172.97   240.3  2172.3     255 2168.06   263.1 2166.88     298 2166.52
   308.9 2164.58   322.6  2166.8   322.6 2166.81   336.4 2166.89   345.6 2170.45
   363.8 2175.05   381.3 2180.74   401.5 2188.42   411.1 2192.96   423.5 2196.14
   439.7 2197.88   450.7 2202.19   462.3  2204.8   477.9 2210.69 482.009 2211.51
#Mann= 4 ,-1 , 0
       0      .1       0  196.17     .06       0     298    .045       0
   322.6    .055       0
Bank Sta=298,322.6
XS Rating Curve= 0 ,0
Exp/Cntr(USF)=0,0
Exp/Cntr=0.3,0.1

Type RM Length L Ch R = 1 ,4093    ,165.9,171.6,160.8
XS GIS Cut Line= 4
2488822.10217152653022.884308015 2488635.6197657653148.820478183
2488499.99619783653252.9600035152488429.76256446653315.928088599
#Sta/Elev= 30
       0 2273.87    19.7 2266.48    71.6 2237.04    90.9 2227.07   116.5  2215.5
     144 2204.87   160.9 2200.68   185.8 2192.27   221.3 2181.97   227.1 2179.08
  233.812173.923   238.5 2172.35   256.4  2171.4   266.5 2165.91   271.5  2164.3
  298.492162.543   311.9 2160.59   321.9 2162.72   341.2 2162.12  346.622163.477
   377.4 2174.24   401.1 2181.38   416.9  2182.8   429.9  2185.4   434.9 2187.18
   440.8 2191.27   443.6 2192.33   446.8 2193.04  462.332193.249 490.345 2194.23
#Mann= 6 ,-1 , 0
       0      .1       0  233.81     .06       0  298.49    .045       0
   321.9     .06       0  346.62    .055       0  462.33      .1       0
Bank Sta=298.49,321.9
XS Rating Curve= 0 ,0
Exp/Cntr(USF)=0,0
Exp/Cntr=0.3,0.1

Type RM Length L Ch R = 1 ,3922    ,131.1,135.1,136.3
XS GIS Cut Line= 4
2488776.08703242652955.0725240792488546.01133693653042.259103426
2488361.95078053653160.9297253152488294.13899659 653216.63226212
#Sta/Elev= 30
       0 2272.24    22.1  2265.2    31.4 2261.48    79.72236.469   108.4 2222.19
   123.7 2215.41  181.062198.854     218 2185.66   233.6 2180.76     246 2173.85
   249.9 2173.04   269.4 2172.03   273.7 2170.71  284.952164.592   295.2 2162.18
  310.822161.449   369.32159.159   390.7 2157.17   394.8 2157.44  400.772159.161
   409.6 2160.92     417 2163.56   431.2 2170.42   439.8 2175.38   457.2 2176.98
   479.5 2186.58  503.92 2191.61   512.2 2192.79   519.9 2196.51552.7979 2207.95
#Mann= 8 ,-1 , 0
       0      .1       0    79.7      .1       0  181.06     .06       0
  284.95      .1       0  310.82    .055       0   369.3    .045       0
  400.77    .055       0  503.92      .1       0
Bank Sta=369.3,400.77
XS Rating Curve= 0 ,0
Exp/Cntr(USF)=0,0
Exp/Cntr=0.3,0.1

Type RM Length L Ch R = 1 ,3787    ,196.2,195.9,181.3
XS GIS Cut Line= 4
2488671.94750709 652875.151493012488514.52729438652942.963276947
2488291.71714716653037.4154045732488197.26501954653090.696091952
#Sta/Elev= 30
       0 2252.53    29.7 2239.54    57.9  2225.8   90.11 2212.66   114.5 2203.74
   191.7 2181.76   197.2 2179.85   205.9 2174.34   210.3 2173.44   229.2 2172.72
   244.4 2164.93   262.7 2159.84  294.722157.795   301.5 2157.93  309.092156.595
   314.5 2154.85   318.9 2154.61   329.5 2156.62   336.3 2157.88   362.3 2155.91
   375.4 2158.68   386.4 2163.19   393.9 2167.23   405.8 2169.05   418.1  2176.4
   432.9 2181.32   483.4  2195.2  502.242202.012     515 2204.51521.8516 2207.89
#Mann= 6 ,-1 , 0
       0      .1       0   90.11     .06       0  294.72    .055       0
  309.09    .045       0   329.5    .055       0  502.24      .1       0
Bank Sta=309.09,329.5
XS Rating Curve= 0 ,0
Exp/Cntr(USF)=0,0
Exp/Cntr=0.3,0.1

Type RM Length L Ch R = 1 ,3591    ,165.2,163.1,151.2
XS GIS Cut Line= 4
2488565.38613234652720.1531297272488400.70037135652785.543064237
2488240.85830921652867.8859447312488153.67172986652906.635535552
#Sta/Elev= 30
       0 2241.97    15.8 2234.42    31.9  2227.6    58.8 2219.06      76 2213.07
   114.7 2202.02   148.9  2193.7   155.1  2191.8   166.4 2187.28   183.9 2175.86
   188.6 2174.65   203.4 2173.73   206.4 2172.97  207.862171.762   210.9 2169.15
   215.7  2163.8   223.8 2156.53   228.9 2153.66  231.152152.903   237.9 2151.18
   242.4 2150.84  255.652152.904   300.9 2153.61  315.942154.843   360.9 2161.93
   372.4 2164.37     390 2166.47   398.7 2170.13  419.332176.809452.4075 2187.74
#Mann= 6 ,-1 , 0
       0      .1       0  207.86     .06       0  231.15    .045       0
  255.65     .06       0  315.94    .055       0  419.33      .1       0
Bank Sta=231.15,255.65
XS Rating Curve= 0 ,0
Exp/Cntr(USF)=0,0
Exp/Cntr=0.3,0.1

Type RM Length L Ch R = 1 ,3428    ,138,140.7,143.8
XS GIS Cut Line= 4
2488524.21469209652567.5766158692488298.98269544652649.919496363
2488160.93727814652751.6371722692488076.17254822652836.401902189
#Sta/Elev= 30
       0 2252.59     5.8 2251.25      33 2240.82    52.7 2231.89    86.7 2215.26
   116.6 2202.24   129.3 2198.07   163.4 2190.24  192.882180.242   218.8 2172.74
   227.3 2167.87   231.5 2166.12     250 2165.72     255 2164.62   268.4 2152.41
     275 2149.56   279.9 2149.44   289.8 2151.22   314.6 2150.94   320.8 2149.01
   330.8 2150.89   362.8 2151.05  373.352153.219   394.1 2156.33   432.1 2165.54
   443.4 2166.67     471 2177.65   494.3 2187.79     517  2196.1531.1605 2202.93
#Mann= 5 ,-1 , 0
       0      .1       0  192.88     .06       0   314.6    .045       0
   330.8     .06       0  373.35    .055       0
Bank Sta=314.6,330.8
XS Rating Curve= 0 ,0
Exp/Cntr(USF)=0,0
Exp/Cntr=0.3,0.1

Type RM Length L Ch R = 1 ,3287    ,199.6,204.1,193.1
XS GIS Cut Line= 4
2488456.40290815652482.8118859482488248.12385749652543.358121606
 2488093.1254942652608.7480561162487996.25151715652669.294291774
#Sta/Elev= 30
       0 2244.62    14.2 2236.99    30.4 2227.07    51.7 2215.74    72.5 2205.88
    98.2 2195.82   126.7 2185.17   197.5  2165.1   201.7 2162.76   205.8 2159.51
     210 2158.39   223.7 2158.45   227.1 2157.57   231.4 2155.06  237.562152.396
   248.1 2149.23   253.1 2148.68   266.2 2149.71   290.9 2149.15   325.5 2149.28
  339.772149.617   348.6 2152.89     366 2158.01   397.4 2165.59   406.8 2168.68
     421 2170.75     442 2177.51   463.9 2183.39   472.6 2186.39499.3664 2198.55
#Mann= 5 ,-1 , 0
       0      .1       0  237.56     .06       0   290.9    .045       0
   325.5     .06       0  339.77    .055       0
Bank Sta=290.9,325.5
XS Rating Curve= 0 ,0
Exp/Cntr(USF)=0,0
Exp/Cntr=0.3,0.1

Type RM Length L Ch R = 1 ,3083    ,154.9,152.2,143.6
XS GIS Cut Line= 4
2488374.06002766652289.0639318432488223.90536323652354.453866354
2488059.21960224652417.4219514382487923.59603436652485.233735374
#Sta/Elev= 30
       0 2256.83    21.1 2248.56    51.6  2232.9    60.3 2227.31    84.7 2209.89
     104 2197.63   134.5 2180.73   156.3  2170.3     165 2163.36   169.3 2160.81
  190.732158.487     195 2156.61   203.6 2150.78   207.8 2149.08  226.422145.444
   232.2 2144.04   237.8 2143.61   250.7 2145.38   263.5 2144.78  292.162146.923
   306.3 2149.65   319.2 2153.31   338.4 2156.08     354 2160.15   370.2 2161.67
   389.8 2161.31   394.3 2161.86     439 2171.01   474.8 2176.24491.7201 2180.09
#Mann= 5 ,-1 , 0
       0      .1       0  190.73     .06       0  226.42    .045       0
   250.7     .06       0  292.16    .055       0
Bank Sta=226.42,250.7
XS Rating Curve= 0 ,0
Exp/Cntr(USF)=0,0
Exp/Cntr=0.3,0.1

Type RM Length L Ch R = 1 ,2931    ,184.6,185.2,184.8
XS GIS Cut Line= 4
 2488277.1860506652146.1748156912488102.81289191652235.783244464
2487972.03302289652313.2824261062487880.00274469652381.094210043
#Sta/Elev= 30
       0 2253.07    14.2  2246.4    65.7 2214.83   124.2  2181.9   132.8 2174.64
   142.2 2168.25   146.7 2166.43   169.1 2165.44   173.6 2163.44   186.5 2155.77
   191.6  2153.6   215.9 2145.18  223.092143.546  231.452142.081   241.4 2140.63
   264.9  2142.2   270.5 2142.64   280.1 2141.26   284.5  2141.6   288.9 2142.59
   297.6 2146.04   303.5 2147.73  329.792152.666   355.9 2157.41   384.4 2161.56
     398  2162.8   409.3  2165.7     425 2168.48     449 2174.49462.3836 2177.02
#Mann= 5 ,-1 , 0
       0      .1       0  223.09     .06       0  231.45    .045       0
   264.9     .06       0  329.79    .055       0
Bank Sta=231.45,264.9
XS Rating Curve= 0 ,0
Exp/Cntr(USF)=0,0
Exp/Cntr=0.3,0.1

Type RM Length L Ch R = 1 ,2745    ,90.2,90.1,90.1
XS GIS Cut Line= 4
 2488185.1557724 652015.394946672488025.31371027652073.519332902
2487870.31534698652163.1277616752487754.06657452652230.939545612
#Sta/Elev= 30
       0  2247.9    19.6 2239.06    35.8 2230.54    83.4 2200.57    98.2 2189.38
   127.3 2173.03   138.8 2163.93     143 2162.41   160.7 2160.71   164.3 2159.28
     173 2153.04   177.7 2150.53   200.8 2140.05     210 2137.34   222.7 2136.49
   233.1  2135.5  247.072137.055   249.22137.204     261 2137.48   274.7 2138.81
   293.2 2142.14   316.4 2147.72  355.472154.909   367.1 2154.41   385.7 2157.37
   413.5 2160.05     432 2163.59   445.9  2165.2     469 2172.26483.7005 2177.95
#Mann= 5 ,-1 , 0
       0      .1       0   222.7    .045       0  247.07      .1       0
   249.2     .06       0  355.47    .055       0
Bank Sta=222.7,247.07
XS Rating Curve= 0 ,0
Exp/Cntr(USF)=0,0
Exp/Cntr=0.3,0.1

Type RM Length L Ch R = 1 ,2655    ,63.5,64.4,64.9
XS GIS Cut Line= 4
2488124.60953675651933.0520661762487986.56411945651991.176452407
2487865.47164813652063.8319351962487734.69177911652143.752966265
#Sta/Elev= 30
       0 2247.19       2 2245.91     8.9 2239.01    19.4 2232.01    23.7    2227
    28.1 2220.46    36.7  2212.9    67.1 2193.66    88.3 2181.53   119.2 2168.35
     125 2165.39   134.2 2159.41   137.2 2158.54   152.4 2157.89   158.2 2156.42
   172.9 2147.46  202.412134.793  209.122132.488   219.4 2130.39  227.822132.489
   236.9 2134.08   257.3 2134.78   280.2  2138.7   296.9  2140.2   309.42142.754
   338.9 2147.85  355.232149.932   373.6 2152.95   382.5 2153.51444.2669 2166.65
#Mann= 6 ,-1 , 0
       0      .1       0  202.41     .06       0  209.12    .045       0
  227.82     .06       0   309.4      .1       0  355.23    .055       0
Bank Sta=209.12,227.82
XS Rating Curve= 0 ,0
Exp/Cntr(USF)=0,0
Exp/Cntr=0.3,0.1

Type RM Length L Ch R = 1 ,2591    ,96.4,95.8,95.2
XS GIS Cut Line= 4
2488124.60953675651870.0839810922487988.98596887651925.786517897
2487838.83130444651998.442000686 2487715.3169837652003.285699539
#Sta/Elev= 30
       0 2256.32    20.4    2247    35.8 2238.37    66.9 2215.96    79.9 2207.63
    88.5 2201.28   101.5 2192.99   123.1 2180.58   144.7  2169.9   158.1 2164.22
   167.1 2157.23   171.3 2155.97   189.1 2155.19   193.5 2153.25  211.042142.216
   215.8 2138.44     221 2133.23   224.6    2131  230.052128.875     239 2126.81
   246.9 2127.38  254.042128.875   264.6 2130.27   298.9 2131.31  314.642134.351
   349.62138.179     364 2139.49   393.6  2145.6  414.692148.667437.0352 2151.56
#Mann= 7 ,-1 , 0
       0      .1       0  211.04     .06       0  230.05    .045       0
  254.04     .06       0  314.64      .1       0   349.6    .055       0
  414.69      .1       0
Bank Sta=230.05,254.04
XS Rating Curve= 0 ,0
Exp/Cntr(USF)=0,0
Exp/Cntr=0.3,0.1

Type RM Length L Ch R = 1 ,2495    ,154.9,157.6,159.2
XS GIS Cut Line= 4
2488056.79775281651787.7411005972487918.75233551651853.131035107
2487773.44136993651928.2083673232487695.94218829651952.426861586
#Sta/Elev= 30
       0 2254.84    11.1  2250.1    21.9 2243.38    24.9 2240.45    35.4 2225.81
      46  2216.1    59.8 2201.25      67 2195.67    99.6 2175.75   112.9 2169.44
   142.1 2158.89   152.8 2152.45  156.992151.741   170.8 2151.47   175.3 2150.67
   185.9 2143.77   197.8 2138.58  220.432126.889   224.8  2125.1   228.3 2124.85
   238.3 2126.62  261.492126.789   281.7 2126.48   290.6 2127.36   296.6  2128.9
   314.8 2137.14   348.5 2139.26     3642144.887   373.6 2147.74397.5046 2152.74
#Mann= 6 ,-1 , 0
       0      .1       0  156.99     .06       0  220.43    .045       0
   238.3     .06       0  261.49    .055       0     364      .1       0
Bank Sta=220.43,238.3
XS Rating Curve= 0 ,0
Exp/Cntr(USF)=0,0
Exp/Cntr=0.3,0.1

Type RM Length L Ch R = 1 ,2337    ,66.1,68.1,69.8
XS GIS Cut Line= 4
2488015.62631256651671.4923281342487872.73719641651732.038563792
2487705.62958599651773.2100040392487654.77074804651804.694046581
#Sta/Elev= 30
       0 2251.99      49  2236.3    53.1  2232.4    61.8  2218.4    70.4 2211.35
    83.5 2204.49    88.7 2199.06    97.9 2185.63   105.2 2177.81   111.2 2172.82
   121.5 2166.98     140 2157.51   165.5 2149.14   169.6 2146.67   173.7 2142.67
   177.8 2141.27   194.3 2140.37   206.7 2132.46   214.9 2128.84   225.3  2125.6
  232.752124.544   247.9 2124.45  253.952122.581   264.3 2119.95  270.832122.579
   276.7 2124.82   309.7 2125.35  332.792130.921   368.3 2141.39387.1075 2143.35
#Mann= 5 ,-1 , 0
       0      .1       0  232.75     .06       0  253.95    .045       0
  270.83     .06       0  332.79      .1       0
Bank Sta=253.95,270.83
XS Rating Curve= 0 ,0
Exp/Cntr(USF)=0,0
Exp/Cntr=0.3,0.1

Type RM Length L Ch R = 1 ,2269    ,82,79.5,75.7
XS GIS Cut Line= 4
 2487998.7536104651579.7659850142487795.91796899651688.393603401
2487738.23958754651691.2775224732487634.41850094 651729.72977677
#Sta/Elev= 30
       0 2241.91     9.1 2239.36    28.9 2236.24    49.6 2229.34    96.9 2211.21
   108.9 2204.02   127.1 2191.57   131.6 2187.22   136.1  2178.4   140.7 2172.15
   149.7 2164.99   158.9 2159.53   188.5 2144.87   195.1 2139.02   199.7 2136.04
   217.8 2135.22   222.3  2133.3   226.9  2129.9   226.9 2129.88   226.9 2129.87
   226.9 2129.86   239.3 2123.55   247.3 2121.31   255.7 2120.22   263.3 2118.95
   271.3 2120.26   279.4 2121.69   321.4 2124.06   344.3 2127.98   398.6 2142.08
#Mann= 5 ,-1 , 0
       0      .1       0   226.9     .06       0   255.7    .045       0
   271.3     .06       0   344.3    .055       0
Bank Sta=255.7,271.3
XS Rating Curve= 0 ,0
Exp/Cntr(USF)=0,0
Exp/Cntr=0.3,0.1

Type RM Length L Ch R = 1 ,2190    ,40.1,40,39.7
XS GIS Cut Line= 4
2488003.51706543651526.1813625552487836.40945502651581.883899361
2487666.87999517651644.8519844452487599.06821124651686.023424692
#Sta/Elev= 30
       0 2257.14   41.25 2242.04    58.1 2235.06    70.7 2232.91    89.4 2227.44
    97.8 2226.05   118.9 2220.73   124.5 2218.71   131.5 2215.17   152.6 2201.37
   169.5 2189.19   173.7 2183.36   177.9 2174.59   181.3 2168.75   187.6 2161.22
   196.9 2148.71   203.5 2141.46   216.3 2130.73   220.6 2128.78   237.7 2128.14
  242.892126.723  253.342119.698   259.1 2117.78   263.3 2117.87  271.582119.697
     323  2121.3  344.122124.247   371.2 2127.44     418 2138.34436.3245  2141.9
#Mann= 6 ,-1 , 0
       0      .1       0   41.25      .1       0  242.89     .06       0
  253.34    .045       0  271.58     .06       0  344.12      .1       0
#XS Ineff= 2 , 0
             203 2121.18     321         2121.18
Permanent Ineff=
       F       F
Bank Sta=253.34,271.58
XS Rating Curve= 0 ,0
Exp/Cntr(USF)=0,0
Exp/Cntr=0.5,0.3

Type RM Length L Ch R = 1 ,2150    ,56.9,56.5,55.9
XS GIS Cut Line= 4
2487976.29897622651493.973726185 2487799.0244449651551.702896328
2487634.52185387651617.0952306492487574.23829567651667.161236614
#Sta/Elev= 30
       0  2255.7    27.3 2244.02    49.6 2235.42    59.1 2230.95    68.9 2229.32
    94.2 2221.19   119.4 2211.03   128.9 2206.49   145.1 2197.17   148.9 2194.49
   161.5 2182.25   169.9 2175.45   182.8 2158.91   186.7 2152.01   195.3 2131.23
   199.7    2126     204 2124.84   212.6 2125.12   225.5 2123.91   229.8 2122.54
   235.3 2119.67   238.4 2118.34     247 2116.81   251.3 2117.17   258.52119.162
   281.4 2120.15   298.7 2119.87   312.3 2121.66   363.5 2127.77   441.8 2142.67
#Mann= 5 ,-1 , 0
       0      .1       0   161.5     .06       0   235.3    .045       0
   258.5     .06       0   312.3    .055       0
#XS Ineff= 2 , 0
             2202121.114     275        2121.114
Permanent Ineff=
       F       F
Bank Sta=235.3,258.5
XS Rating Curve= 0 ,0
Exp/Cntr(USF)=0,0
Exp/Cntr=0.5,0.3

Type RM Length L Ch R = 1 ,2093    ,83.7,82.5,80.8
XS GIS Cut Line= 4
 2487889.4497822651452.5926396222487755.59984789 651506.23478887
2487606.93446283651574.1815112512487533.36808672651594.105738114
#Sta/Elev= 30
       0 2233.29    11.5 2228.69    19.2 2224.52    28.5 2223.18    37.4 2218.35
    54.6 2210.98    67.6 2207.03    83.8 2203.14    97.7 2196.84     102 2192.77
   119.3 2173.09   123.8 2164.41   127.9 2157.87   130.2 2153.34   133.1 2147.36
   140.8 2129.36   145.1 2122.87   148.4 2121.91   167.1 2120.58   171.5 2119.73
   174.92117.963   180.3 2115.91   184.3 2115.79   193.9  2117.8   202.3 2118.44
   215.5 2117.69   280.5  2124.2   299.3  2126.7   353.4 2136.37   383.9 2140.38
#Mann= 5 ,-1 , 0
       0      .1       0   148.4     .06       0   174.9    .045       0
   193.9     .06       0   280.5    .055       0
Bank Sta=174.9,193.9
XS Rating Curve= 0 ,0
Exp/Cntr(USF)=0,0
Exp/Cntr=0.5,0.3

Type RM Length L Ch R = 1 ,2011    ,88.8,89,89
XS GIS Cut Line= 4
2487829.56369149651361.549441883 2487700.7486396651438.453950475
2487643.07025816651476.906204772 2487524.8295762651549.004181577
#Sta/Elev= 30
       0 2227.18    12.6  2221.7    21.9 2216.81      26 2215.07    35.1 2213.71
    45.2 2209.42    59.2 2204.88      73 2198.89    82.5 2193.64    99.3 2181.54
   105.8 2176.17     111  2170.1   115.1 2164.34   122.6 2156.95   124.4 2154.84
   128.5  2146.8   133.7 2137.68     143 2123.55     146 2120.65   147.7 2119.56
   148.9 2119.36   166.9 2118.99   176.5 2115.85   186.9 2115.22   195.1 2113.94
   206.6 2115.61   247.2  2118.1   282.1 2124.65   317.1 2131.52   357.8 2137.69
#Mann= 5 ,-1 , 0
       0      .1       0   166.9     .06       0   186.9    .045       0
   206.6     .06       0   282.1    .055       0
Bank Sta=186.9,206.6
XS Rating Curve= 0 ,0
Exp/Cntr(USF)=0,0
Exp/Cntr=0.3,0.1

Type RM Length L Ch R = 1 ,1922    ,142.6,138.2,132.7
XS GIS Cut Line= 4
2487773.44136993651317.9023118932487686.25479058651344.542655582
2487548.20937329651431.7292349292487482.81943877651509.228416571
#Sta/Elev= 30
       0 2215.57    11.2  2214.4    22.2 2211.39    44.4 2204.33    58.1 2199.01
    63.8 2196.12    78.1    2185    86.2 2176.97    95.3 2171.59    98.3 2167.51
     100 2164.54   103.1 2157.32   114.2 2128.43     118 2120.43     119 2118.95
   123.7 2116.72   142.6 2116.02  150.462114.632  154.672112.881   156.8 2111.95
     163 2111.05  175.62 2112.88   207.9 2113.92   222.9 2113.22  259.252119.004
   280.4 2124.29   308.8 2133.36   314.5 2134.35   328.7 2135.22355.8387 2139.56
#Mann= 5 ,-1 , 0
       0      .1       0  150.46     .06       0  154.67    .045       0
  175.62     .06       0  259.25    .055       0
Bank Sta=154.67,175.62
XS Rating Curve= 0 ,0
Exp/Cntr(USF)=0,0
Exp/Cntr=0.3,0.1

Type RM Length L Ch R = 1 ,1784    ,116.5,119.1,119.2
XS GIS Cut Line= 4
2487676.56739288 651175.013195742487555.47492156651245.246829103
2487470.71019164651368.7611498452487427.11690197651436.572933782
#Sta/Elev= 30
       0 2219.88    15.9 2215.82    39.6 2206.15      51  2200.7    66.8 2189.98
    77.22178.934    80.7 2175.47    87.5 2170.63      90 2168.39      92 2165.69
    94.9 2160.84   106.6 2135.65   109.5 2130.25   127.1 2114.26   151.7 2113.29
   166.2 2111.77  186.942106.844   190.5  2105.9   200.2  2105.3   204.9  2105.7
   210.7 2107.08   214.8 2107.22     228 2106.44   253.9 2108.89   263.3 2108.75
   268.3 2109.52   292.3 2116.23   344.6 2133.24   354.1 2135.66370.4041 2138.35
#Mann= 4 ,-1 , 0
       0      .1       0    77.2     .06       0  186.94    .045       0
   214.8    .055       0
Bank Sta=186.94,214.8
XS Rating Curve= 0 ,0
Exp/Cntr(USF)=0,0
Exp/Cntr=0.3,0.1

Type RM Length L Ch R = 1 ,1665    ,105.3,106.1,106.7
XS GIS Cut Line= 4
2487586.95896411651087.8266163932487465.86649279651187.122442872
2487366.57066631651291.2619682032487298.75888238651373.604848698
#Sta/Elev= 30
       0 2212.83    16.5 2210.69    26.1 2207.58    31.3 2203.55    41.7 2190.21
      45 2187.12    57.2 2180.16    59.2 2178.42    62.4  2174.8    64.9 2169.72
    76.2 2142.87    81.9 2131.14    87.6 2121.34    90.4  2117.4    93.4 2114.02
  111.242111.671   118.4 2110.39   137.3 2109.24   178.4 2108.69  194.69 2102.99
     206 2101.02  219.05 2102.99   226.5 2103.83  232.922103.662   265.5 2103.81
   288.9 2108.34   317.2 2116.71     337 2123.91   356.8 2130.09 407.161  2144.1
#Mann= 5 ,-1 , 0
       0      .1       0  111.24     .06       0  194.69    .045       0
  219.05     .06       0  232.92    .055       0
Bank Sta=194.69,219.05
XS Rating Curve= 0 ,0
Exp/Cntr(USF)=0,0
Exp/Cntr=0.3,0.1

Type RM Length L Ch R = 1 ,1558    ,93.9,93.5,89.3
XS GIS Cut Line= 4
2487526.41272845651000.6400370462487415.00765484651095.092164672
2487281.80593639651218.6064854142487226.10339959651305.793064761
#Sta/Elev= 30
       0 2203.86      22 2197.04    25.8 2194.39    36.3 2181.72    41.5 2177.69
    55.3  2169.6   59.692165.792    69.5 2154.24    80.8 2131.84    83.7 2126.96
    86.5 2123.65    89.3 2121.48    92.2  2120.8  104.232120.595   114.9 2119.03
   129.1 2108.21   133.4 2106.24   157.4 2105.52   174.4    2102  204.592100.212
     214 2098.34  225.012100.212   245.8 2101.33   275.2    2101   281.42101.967
     328  2114.3   356.2 2118.98   370.7  2122.4   414.1 2138.84431.1721 2143.99
#Mann= 6 ,-1 , 0
       0      .1       0   59.69     .12       0  104.23     .06       0
  204.59    .045       0  225.01     .06       0   281.4    .055       0
Bank Sta=204.59,225.01
XS Rating Curve= 0 ,0
Exp/Cntr(USF)=0,0
Exp/Cntr=0.3,0.1

Type RM Length L Ch R = 1 ,1465    ,147.5,151.7,110.8
XS GIS Cut Line= 4
2487453.75724566650918.2971565522487344.77402148651024.858531309
2487230.94709844 651155.638400332487180.08826049651237.981280825
#Sta/Elev= 30
       0 2179.94    15.4 2175.18      18 2172.51      28 2158.71    30.8 2156.11
    43.4 2149.94    54.6 2139.33    71.3  2126.1    78.9 2122.72   84.992122.013
    92.4 2121.44   104.4 2121.86  112.382120.988   116.1 2119.92   138.2 2110.12
   149.6 2103.19   176.3 2101.72     186 2100.26   198.2 2099.63   206.3 2097.89
     212 2097.19   217.7 2098.09     229 2099.52  242.942098.979   266.5 2098.24
   282.4 2096.05   299.9 2097.75   334.3 2111.75  375.582123.506422.5838 2139.33
#Mann= 7 ,-1 , 0
       0      .1       0   84.99     .12       0  112.38     .06       0
   206.3    .045       0   217.7     .06       0  242.94      .1       0
  375.58    .055       0
Bank Sta=206.3,217.7
XS Rating Curve= 0 ,0
Exp/Cntr(USF)=0,0
Exp/Cntr=0.3,0.1

Type RM Length L Ch R = 1 ,1313    ,160.1,162.4,163.8
XS GIS Cut Line= 4
2487359.30511803650799.6265346622487240.63449614650954.624897946
2487155.86976622651080.5610681142487102.58907884651158.060249756
#Sta/Elev= 30
       0 2160.47     9.1  2156.5    19.2 2148.37    24.3 2145.93    33.8  2139.3
    39.4 2137.14    49.5  2135.2    66.7 2130.04   112.8 2129.29   119.4 2128.56
   130.1 2124.47   139.7 2119.65  160.852115.969   165.3  2114.1   176.8 2112.02
   185.2 2109.24   190.5 2106.85   196.8 2102.86   200.4 2101.56   224.5  2100.6
   237.1 2097.87   301.6 2094.19     312 2093.11   320.7 2094.36   329.3 2096.17
   343.7 2105.81   358.1 2112.29   392.6 2124.27   424.3 2133.93 441.064 2140.03
#Mann= 4 ,-1 , 0
       0      .1       0  160.85     .06       0   301.6    .045       0
   320.7    .055       0
Bank Sta=301.6,320.7
XS Rating Curve= 0 ,0
Exp/Cntr(USF)=0,0
Exp/Cntr=0.3,0.1

Type RM Length L Ch R = 1 ,1151    ,231.7,233.3,235.1
XS GIS Cut Line= 4
2487319.75415012650676.8142955562487124.11626017650872.452185503
2487020.76039378650979.499332833 2486891.5655608651053.324951681
#Sta/Elev= 30
       0 2191.98    27.6 2176.12    41.8 2164.18    48.2 2156.34    55.9 2141.21
    59.5 2136.96   155.7 2132.68   163.4 2131.08   172.6 2126.02   182.4 2123.32
  242.73 2118.86   276.7 2113.33   296.3 2099.38   299.2 2098.53     319 2097.97
   330.3 2093.38   353.5 2093.83  364.532090.506   370.8 2088.62  380.732090.508
   399.6 2104.68   419.1  2115.3   438.2 2119.33   467.5 2121.74  480.942125.433
   496.9 2131.14   514.5 2133.15   524.5 2138.09   552.2 2145.36574.2744 2157.11
#Mann= 5 ,-1 , 0
       0      .1       0  242.73     .06       0  364.53    .045       0
  380.73    .055       0  480.94      .1       0
Bank Sta=364.53,380.73
XS Rating Curve= 0 ,0
Exp/Cntr(USF)=0,0
Exp/Cntr=0.3,0.1

Type RM Length L Ch R = 1 ,918     ,214.6,229.5,242.3
XS GIS Cut Line= 4
2487260.69365504650551.3107435142487042.90807944650665.740452728
2486847.27018949 650806.009128542486747.60560405650853.995780791
#Sta/Elev= 30
       0  2211.3     2.2 2210.09     6.7 2204.29    15.9 2188.77    33.8 2174.35
    56.4 2160.83    78.1 2150.92   128.7 2133.48   155.8  2127.4   164.9 2126.61
   175.9  2122.9   214.1 2116.64   232.2 2111.74   252.7 2103.38   273.62097.952
   304.3 2089.51     325 2089.74   339.7 2087.93   374.2  2087.8  384.512086.512
  391.232084.062     399 2081.72  414.132084.063   438.2 2092.54   467.7 2108.59
     482  2113.4  494.842115.712     545  2136.1   576.1 2145.47  597.36 2156.75
#Mann= 6 ,-1 , 0
       0      .1       0   273.6     .06       0  384.51    .055       0
  391.23    .045       0  414.13    .055       0  494.84      .1       0
Bank Sta=391.23,414.13
XS Rating Curve= 0 ,0
Exp/Cntr(USF)=0,0
Exp/Cntr=0.5,0.3

Type RM Length L Ch R = 1 ,688     ,51.7,50.5,50.1
XS GIS Cut Line= 4
2487234.85468844 650499.632810322486906.33068457650625.136362362
2486777.13585159650481.1764056082486596.26308541650647.284048016
#Sta/Elev= 30
       0 2206.03     4.4 2202.93    21.5 2181.61    52.2  2164.2    67.7 2156.59
     111 2139.56   137.1 2130.55   176.1 2118.32   188.5 2116.07  245.86 2100.68
     287 2089.15   308.4 2085.98   346.5 2086.11   392.6 2083.45   410.9  2080.2
  432.852079.888   443.6 2077.97  451.532079.889   460.6 2083.41   478.3 2086.15
   497.4 2087.96   515.9 2087.63  527.562088.481   570.1 2094.16   580.9 2099.51
   652.8 2125.81     695 2142.61   725.1 2156.17   765.6 2177.31790.6863 2192.58
#Mann= 5 ,-1 , 0
       0      .1       0  245.86     .06       0  432.85    .045       0
  451.53     .06       0  527.56      .1       0
#XS Ineff= 2 , 0
             410 2079.79     473         2079.79
Permanent Ineff=
       F       F
Bank Sta=432.85,451.53
XS Rating Curve= 0 ,0
Exp/Cntr(USF)=0,0
Exp/Cntr=0.5,0.3

Type RM Length L Ch R = 1 ,638     ,164,156.3,143.8
XS GIS Cut Line= 4
2487227.47212656 650407.350786762486926.91849688650575.145566036
2486800.80558448 650437.193408062486575.93002264650628.047984753
#Sta/Elev= 30
       0 2223.38    37.5 2213.18    41.4 2208.22    51.2 2188.85    55.8 2181.46
    69.5 2171.39    78.7 2162.53    88.4 2157.05   144.2 2135.74   188.3 2120.85
   234.5 2109.06   269.8 2097.46  291.39 2093.14  366.282084.302  388.06 2081.93
   412.5 2078.95     421 2076.28   426.6 2075.26   435.1 2076.18   458.4 2077.39
   545.1    2076   549.6 2076.43  555.572079.718     582 2091.12   601.8  2094.9
     623 2105.27   672.9 2123.63   743.8 2152.89   790.9 2176.75826.0783 2199.33
#Mann= 7 ,-1 , 0
       0      .1       0  291.39     .06       0  366.28      .1       0
  388.06     .06       0     421    .045       0   435.1     .06       0
  555.57      .1       0
Bank Sta=421,435.1
XS Rating Curve= 0 ,0
Exp/Cntr(USF)=0,0
Exp/Cntr=0.5,0.3

Type RM Length L Ch R = 1 ,481     ,160.3,159.8,158.9
XS GIS Cut Line= 4
2487145.46532287 650211.289879412486879.47083947650338.566809639
2486743.61344204650421.5113259682486550.55292989650598.840981569
#Sta/Elev= 30
       0 2217.73    54.7 2189.22    63.9  2183.5    91.7 2168.72   163.7 2126.28
   193.7 2112.62   224.7 2103.29     240 2099.56   251.3 2097.36   286.8 2092.87
  311.122087.762  378.672071.223   389.5  2069.3   394.1 2069.61  398.552071.222
   406.2 2074.77  418.392075.417     427 2075.47   441.1 2080.72     447 2083.32
   456.1 2089.48   460.7  2091.2     484 2093.16   495.3 2100.16   525.8 2112.48
   605.7 2141.98   639.7 2157.93   656.2 2166.96   692.6 2189.26716.1946 2205.31
#Mann= 5 ,-1 , 0
       0      .1       0  311.12     .06       0  378.67    .045       0
  398.55     .06       0  418.39      .1       0
Bank Sta=378.67,398.55
XS Rating Curve= 0 ,0
Exp/Cntr(USF)=0,0
Exp/Cntr=0.3,0.1

Type RM Length L Ch R = 1 ,321     ,179.2,176.2,166.6
XS GIS Cut Line= 4
 2487070.7501298650037.5913268742486817.69108325650186.680377557
2486678.41052274650280.8418832522486480.27902117650514.283949454
#Sta/Elev= 30
       0 2235.24    34.1 2220.83    50.6 2212.05    60.4 2204.93      74 2190.92
    83.6  2184.2    92.9 2171.97      98 2167.42   128.6 2147.78     168 2128.11
   207.4 2111.94   241.4 2101.32  379.322067.506  380.242067.278     389  2065.4
  401.452067.278   422.7 2071.78   457.3 2070.75  493.962083.425   522.6 2087.35
     534 2093.74   627.2 2129.14   661.7 2146.14   708.6 2173.72   720.9 2192.14
   727.1 2199.06   747.8 2214.06  755.062223.216     761 2231.05768.0231 2235.37
#Mann= 6 ,-1 , 0
       0      .1       0  379.32     .06       0  380.24    .045       0
  401.45     .06       0  493.96      .1       0  755.06      .1       0
Bank Sta=380.24,401.45
XS Rating Curve= 0 ,0
Exp/Cntr(USF)=0,0
Exp/Cntr=0.3,0.1

Type RM Length L Ch R = 1 ,145     ,147.8,145.2,139.6
XS GIS Cut Line= 4
2486743.14655791649959.1234054612486660.75524042650063.093401333
2486541.09166027650259.2632048642486474.39392707650363.233200735
#Sta/Elev= 30
       0 2116.52   54.862102.063    81.4 2093.06    96.7 2082.99   106.9 2081.91
   117.1 2076.56   127.3 2073.62   160.2 2069.03   165.2 2066.73  170.932062.692
   174.9 2060.87  199.45 2062.69   207.4    2064   216.8 2064.42   228.7 2068.13
   249.6 2068.04     262 2075.54   270.8 2077.51  313.772077.708     329 2078.51
   343.3 2082.71   352.6 2084.06   375.5 2091.65   404.8 2103.18   421.8 2113.08
   430.5 2118.94   436.3  2123.2   452.3 2136.83   479.7  2156.3485.9693 2161.35
#Mann= 5 ,-1 , 0
       0      .1       0   54.86      .1       0  170.93    .045       0
  199.45     .06       0  313.77      .1       0
Bank Sta=170.93,199.45
XS Rating Curve= 0 ,0
Exp/Cntr(USF)=0,0
Exp/Cntr=0.3,0.1
